HEC-RAS study BEAVERCK.prj: BEAVERCK

--- BEAVERCK.g01 (geometry) --- (continued)

Type RM Length L Ch R = 1 ,34562   ,65.3,64.3,66.5
XS GIS Cut Line= 2
2228915.99177662 407249.677871022229446.42676554406785.666222633
#Sta/Elev= 30
       0 2482.87      19 2479.42    37.4 2472.95    42.8 2472.12    74.6 2470.11
   170.9  2467.1   207.4 2466.53   244.7 2464.04   335.1 2463.88   374.7 2464.84
   409.5 2463.95   441.3 2465.57     452 2465.26   473.2 2465.71   489.2 2467.55
   498.9 2463.91   505.1 2463.22   510.7 2463.59   521.1 2462.81   533.4 2463.87
   544.8 2465.52   595.5 2466.88   611.4 2472.35   620.4 2472.52   638.7 2471.45
   641.1 2472.21   653.9 2478.62   666.6 2483.28   680.8 2489.47   704.7 2498.68
#Mann= 10 ,-1,0
       0     .06       0      80      .1       0     100     .06       0
     230     .05       0     360     .06       0     380     .05       0
     490     .07       0   498.9    .045       0   533.4     .07       0
     680      .1       0
#XS Ineff= 2 , 0
          489.81  2468.4  541.89          2468.4
Permanent Ineff=
       F       F
Bank Sta=498.9,533.4
XS Rating Curve= 0 ,0
Exp/Cntr(USF)=0,0
Exp/Cntr=0.5,0.3

Type RM Length L Ch R = 1 ,34498   ,139.9,146.9,148.6
XS GIS Cut Line= 2
2228942.70529814407298.3068958692229486.06036225406839.934252615
#Sta/Elev= 30
       0 2471.46    41.6 2471.07    64.7 2469.49   117.1 2467.99   263.6 2465.45
     295 2463.88   328.3 2463.45   336.8 2464.28     351 2462.39     368 2465.48
   413.4 2465.07   479.4 2465.99   488.6 2465.11   493.8 2463.39   498.6 2462.22
   504.3 2463.47   509.5 2463.24     520 2461.62   525.2 2462.48     527 2463.49
   535.5 2467.45   556.6 2468.46   575.2 2470.74   603.5 2470.99   615.9 2471.85
   634.8 2471.47     649 2478.13   677.9 2489.53   697.9 2497.24   710.9 2501.39
#Mann= 9 ,-1,0
       0     .05       0      10     .06       0     310     .05       0
     320     .06       0     450     .05       0     470     .07       0
   493.8    .045       0     527     .07       0     700      .1       0
#XS Ineff= 2 , 0
          491.93  2468.4  527.86          2468.4
Permanent Ineff=
       F       F
Bank Sta=493.8,527
XS Rating Curve= 0 ,0
Exp/Cntr=0.5,0.3

Type RM Length L Ch R = 1 ,34351   ,168.1,168.7,169.5
XS GIS Cut Line= 3
2228949.54868636407312.4820151642229084.57530055407295.592412404
2229549.38734553406992.358100821
#Sta/Elev= 30
       0 2471.33   145.2 2468.24   245.4 2465.19   287.8 2463.44     311 2463.18
   321.9  2462.4   350.5 2461.59   374.8 2462.47   383.2 2462.27   391.9 2460.63
   396.7 2460.29   417.4 2462.14   465.1 2462.39   469.62461.891   474.7 2460.54
   479.5 2459.99   484.2 2460.54   490.52462.129   499.2 2464.03   536.8 2464.66
   588.4  2466.4     600 2467.52   608.4 2470.88   613.2 2471.54   641.9    2472
   649.1 2475.42   660.7 2482.94   670.5 2487.75   683.8 2496.37   691.1 2500.15
#Mann= 10 ,-1,0
       0     .05       0      40     .06       0  136.08     .05       0
  316.08     .06       0  376.08     .05       0   469.6    .045       0
   490.5     .05       0  496.08      .1       0  606.08     .07       0
  676.08     .06       0
Bank Sta=469.6,490.5
XS Rating Curve= 0 ,0
Exp/Cntr(USF)=0,0
Exp/Cntr=0.3,0.1

Type RM Length L Ch R = 1 ,34182   ,321,318.9,313
XS GIS Cut Line= 4
2229086.75766763407320.4792887472229370.15870632407294.639782277
2229440.17543353407257.130821273 2229754.4171735 407026.24232798
#Sta/Elev= 30
       0 2468.79    33.6 2467.98    45.6 2467.15    81.8 2467.08   125.9 2465.44
     146 2465.74   182.2 2465.14   250.5 2462.44   309.6 2461.28   323.2 2460.25
   331.5 2458.73   336.8 2458.49     3492460.108   355.1 2460.62   372.6 2460.13
   433.5  2460.6     445 2461.16   484.1 2465.59   512.9 2468.14   532.8 2472.31
   552.8 2472.09   572.5 2473.38   582.4 2475.65   654.4 2480.92   667.3 2482.68
   710.2  2486.7   721.4 2488.95   730.2 2489.05   741.7 2490.96     754 2491.81
#Mann= 9 ,-1,0
       0     .05       0     100     .07       0     200     .05       0
   323.2    .045       0     349     .05       0  414.01      .1       0
  464.01     .06       0  634.01      .1       0  664.01     .08       0
Bank Sta=323.2,349
XS Rating Curve= 0 ,0
Exp/Cntr(USF)=0,0
Exp/Cntr=0.3,0.1

Type RM Length L Ch R = 1 ,33863   ,201.9,204.2,204.4
XS GIS Cut Line= 3
2229138.80855103407657.3613819892229433.83181231407596.662816271
2229767.65526869 407348.88164433
#Sta/Elev= 30
       0 2481.09    17.7  2478.1   160.7 2464.03     226 2461.75   283.2 2460.85
   368.3  2458.4     394 2458.43   434.6  2457.3   468.3  2457.4   485.5 2456.88
   501.7 2457.42   528.3 2456.75   573.1 2458.22   583.1 2457.87   588.1 2456.85
     593 2455.35     597 2455.01   608.4 2456.72     618 2456.72   622.9 2457.61
   635.9 2456.94   647.8 2458.13   657.1 2462.87   667.8 2470.42   671.3 2471.86
   682.7 2472.44   699.9 2472.04   702.8 2472.84   705.7 2474.41   716.9 2481.91
#Mann= 6 ,-1,0
       0     .08       0      50     .05       0   481.2      .1       0
   588.1    .045       0   608.4      .1       0   641.2     .06       0
Bank Sta=588.1,608.4
XS Rating Curve= 0 ,0
Exp/Cntr(USF)=0,0
Exp/Cntr=0.3,0.1

Type RM Length L Ch R = 1 ,33659   ,211.8,214.2,215.2
XS GIS Cut Line= 3
2229212.45754423 407868.994055162229515.95037282407777.240409308
 2229895.6693072407494.921498992
#Sta/Elev= 30
       0  2503.1    12.2  2497.2    37.3 2487.43    58.2 2480.58    99.1 2471.23
   118.3 2467.52   137.6 2464.59   160.1 2462.22   192.1 2460.21   217.8 2459.39
   417.7 2455.89   541.6 2455.62   565.2 2455.05   581.5  2455.5   618.8 2454.91
   661.3 2456.08   679.2 2455.38   701.1 2453.11   712.7  2455.4   716.1 2456.54
   721.1 2459.35   726.1 2462.86     736 2471.41   737.5 2472.19     741 2473.24
   746.2 2473.76   766.1 2473.58   771.8 2476.15   780.9 2482.15   790.2 2486.99
#Mann= 7 ,-1,0
       0     .08       0      80     .05       0  517.06      .1       0
  647.06     .08       0   679.2    .045       0   712.7     .08       0
  767.06     .06       0
Bank Sta=679.2,712.7
XS Rating Curve= 0 ,0
Exp/Cntr(USF)=0,0
Exp/Cntr=0.3,0.1

Type RM Length L Ch R = 1 ,33445   ,141.2,144.1,141.4
XS GIS Cut Line= 2
 2229359.2633776408062.3825087262230011.42006043407637.492548702
#Sta/Elev= 30
       0 2483.26    48.8 2477.93    65.1  2475.4   105.6 2471.72   134.8 2468.29
   156.1 2466.71   196.8  2461.4   220.7 2459.81   235.7 2457.97   255.9 2456.54
   377.3  2454.9   411.7 2453.82   516.7 2454.69   550.8 2454.15   562.3 2452.71
   578.7 2451.09   585.5 2451.32   595.8 2452.64   650.4 2453.43   654.8 2454.69
   660.6 2457.92   666.4 2459.82   693.3 2464.72     713 2469.26   717.2 2470.91
   727.6  2476.7   736.3 2477.43     756 2476.98   764.9 2481.96   778.4 2486.32
#Mann= 11 ,-1,0
       0      .1       0     150     .05       0     260     .08       0
     330     .05       0     380     .07       0     500     .08       0
     510      .1       0   562.3    .045       0   595.8      .1       0
     620     .06       0     730     .07       0
Bank Sta=562.3,595.8
XS Rating Curve= 0 ,0
Exp/Cntr(USF)=0,0
Exp/Cntr=0.3,0.1

Type RM Length L Ch R = 1 ,33301   ,211.5,212,212
XS GIS Cut Line= 2
2229423.39531524 408194.451720462230083.44900704407735.843010053
#Sta/Elev= 30
       0 2513.57    15.6 2508.38    25.3 2504.51    39.9 2497.82    88.6 2473.41
   100.4 2468.54     113 2465.94   130.8 2464.04   234.7 2455.94   306.1  2453.5
   435.4  2451.8   517.2 2452.49   536.7 2451.98     605 2453.16   626.1 2452.55
   630.9 2451.84   640.2 2450.22   653.6 2449.71   661.2 2450.15   665.4 2451.87
     674 2457.43   702.7 2466.38     720 2470.13   738.3 2474.27   748.7 2475.43
   760.8 2478.93   771.7 2479.39   788.9 2478.82   797.6 2484.04   803.7 2488.69
#Mann= 8 ,-1,0
       0      .1       0     370     .08       0     430     .07       0
     540     .08       0     550      .1       0   630.9    .045       0
   665.4      .1       0     720     .06       0
Bank Sta=630.9,665.4
XS Rating Curve= 0 ,0
Exp/Cntr=0.3,0.1

Type RM Length L Ch R = 1 ,33089   ,395.1,427.1,448.9
XS GIS Cut Line= 2
2229610.53037434408314.6518962472230198.23364994407915.608232462
#Sta/Elev= 30
       0 2469.94    35.8 2460.71   109.4 2454.85   195.2 2450.11   243.7 2448.96
   290.2 2449.41     319 2448.43   365.1 2449.58   385.2 2448.56   393.6  2449.3
     414 2448.92     440 2449.53   460.1 2450.11   471.6 2448.24   485.5 2448.43
   497.5 2449.94   524.2  2450.8   538.7 2450.01   548.3 2448.89   567.7 2448.98
     573 2449.92   582.2 2460.29   583.9 2461.68     587 2463.71   591.8 2465.14
   635.8 2466.72   657.7 2468.44   683.7 2470.96   698.2 2475.45   710.4 2475.68
#Mann= 6 ,-1,0
       0      .1       0     440     .08       0   538.7    .045       0
     573     .08       0     590      .1       0     680     .06       0
Bank Sta=538.7,573
XS Rating Curve= 0 ,0
Exp/Cntr(USF)=0,0
Exp/Cntr=0.3,0.1

Type RM Length L Ch R = 1 ,32662   ,302.6,284.7,245.2
XS GIS Cut Line= 4
2229661.98299575408328.3725952892229904.38201214408354.670601785
2230032.44186986408470.1531520492230372.02917113408259.769100082
#Sta/Elev= 30
       0 2461.39    94.7 2455.04   166.1    2449   231.5 2445.25   245.5 2445.31
   259.6 2446.19   266.92445.899   276.6 2443.36   281.2 2443.02   287.9 2443.69
   295.62445.715   313.4 2445.75   324.3 2446.62   383.6 2444.72     389 2445.62
   392.7 2447.19   399.7 2448.77   416.3 2448.72   433.3 2450.37     463    2452
   477.1 2451.95   486.5 2452.81   509.3 2453.18     543 2452.05   575.9 2452.43
     608 2454.45   681.2 2456.42     703  2458.1   735.9 2458.22   815.7 2461.38
#Mann= 5 ,-1,0
       0      .1       0   266.9    .045       0   295.6     .08       0
  466.26     .12       0  806.26     .06       0
Bank Sta=266.9,295.6
XS Rating Curve= 0 ,0
Exp/Cntr(USF)=0,0
Exp/Cntr=0.3,0.1

Type RM Length L Ch R = 1 ,32377   ,307.6,308.5,310.3
XS GIS Cut Line= 4
2229808.33711885 408718.269126382229870.08026454408667.959896562
2230039.30221938408522.7491650412230386.89326176408294.070847685
#Sta/Elev= 30
       0 2552.32    27.1 2540.52      49 2529.25    63.2 2520.91    83.9 2507.19
    92.9 2500.24   111.5 2486.83   126.9 2473.32   135.1 2465.59   155.3 2442.52
   157.6  2440.8   163.8  2440.2   177.3 2440.28   182.4 2440.93   185.2 2441.96
   188.3 2443.04   198.4 2443.86   227.8 2444.01   280.5 2445.47   315.9 2447.41
   337.2 2447.51   359.3 2448.76   375.5 2450.78   400.1 2450.12   480.6 2453.03
   528.7 2452.98     634 2457.69   662.1 2459.58   682.7 2459.68   718.7 2461.13
#Mann= 5 ,-1,0
       0      .1       0   155.3    .045       0   185.2      .1       0
  342.63     .12       0  692.63     .07       0
#XS Ineff= 2 , 0
                          272.44         2460.38
Permanent Ineff=
       F       F
Bank Sta=155.3,185.2
XS Rating Curve= 0 ,0
Exp/Cntr(USF)=0,0
Exp/Cntr=0.3,0.1

Type RM Length L Ch R = 1 ,32068   ,250.8,249.1,249.1
XS GIS Cut Line= 3
2229959.26480831408982.3925829262230211.95434899408788.016013173
2230561.83217454408383.255391454
#Sta/Elev= 30
       0 2572.07    47.2 2544.73    81.9 2523.19     107 2506.46   117.2 2498.86
   135.6 2486.71   152.7 2474.81   162.6 2467.39   172.7 2460.73   181.2  2454.3
   195.5 2441.87   198.3 2440.16   201.2 2439.35   205.4 2438.72   226.9 2437.95
   244.7 2438.78   251.3 2439.36   258.5 2441.17   268.6 2442.19   397.5 2444.26
     417 2445.59   445.7 2449.05   471.3 2450.93   502.5  2451.1   539.3 2452.03
   658.4 2456.37   692.7 2458.07   793.1 2461.16   845.6 2463.26   853.8 2465.19
#Mann= 7 ,-1,0
       0      .1       0   201.2    .045       0   244.7      .1       0
   408.8     .05       0   598.8      .1       0   708.8     .05       0
   728.8     .06       0
Bank Sta=201.2,244.7
XS Rating Curve= 0 ,0
Exp/Cntr(USF)=0,0
Exp/Cntr=0.3,0.1

Type RM Length L Ch R = 1 ,31819   ,348.4,346,347.5
XS GIS Cut Line= 3
 2230129.6567942 409178.44086747  2230565.185274408803.966243845
2230757.21284314408598.812156865
#Sta/Elev= 30
       0 2525.51    24.4 2513.05    50.8  2497.1    56.6 2493.14    61.3 2488.52
    66.6  2484.3   124.6 2447.53   129.9 2443.02   133.2 2440.99     136 2439.98
   164.4 2438.88   175.7 2437.79   181.4 2436.73     188 2436.53   204.1  2436.6
   209.7  2437.5   224.9 2437.81   240.7 2439.53   260.8 2438.08   272.1 2439.78
   362.9 2440.16   409.5  2441.4   473.5 2441.83   499.2 2442.83     587 2450.71
   666.6 2453.24   722.8 2456.79   818.7 2467.27   841.7 2465.64   855.4 2466.57
#Mann= 5 ,-1,0
       0      .1       0   175.7    .045       0   209.7      .1       0
     310     .05       0  855.39     .06       0
Bank Sta=175.7,209.7
XS Rating Curve= 0 ,0
Exp/Cntr=0.3,0.1

Type RM Length L Ch R = 1 ,31473   ,159.3,165.4,166.7
XS GIS Cut Line= 4
2230220.98408116409316.1522835862230460.95515493409344.384174618
2230675.83121445 409154.603129352230832.67505351408870.715780644
#Sta/Elev= 30
       0 2499.12     7.2 2495.48    15.3 2492.51    43.4 2480.02    59.6 2468.24
    91.8 2451.83   107.9 2449.01   132.1 2446.06   151.5 2442.57   164.3 2441.56
   176.4  2441.5     220 2438.29   267.3 2435.82   315.3 2435.47   331.1 2436.29
   336.6 2434.97   342.5  2433.5   348.2  2433.4     368  2434.9   373.7 2435.56
   395.4 2435.02   413.4 2436.25   424.6 2435.12   476.1 2434.49   492.7 2437.51
   535.5 2437.46   676.2 2443.81     768 2452.48   812.2 2455.19   852.6 2456.66
#Mann= 5 ,-1,0
       0     .12       0      50      .1       0   336.6    .045       0
     368      .1       0  628.31     .05       0
Bank Sta=336.6,368
XS Rating Curve= 0 ,0
Exp/Cntr(USF)=0,0
Exp/Cntr=0.3,0.1

Type RM Length L Ch R = 1 ,31308   ,281.1,285.1,283.3
XS GIS Cut Line= 3
2230330.94450075409584.4837717452230919.63969482  409211.3719814
2231012.63193011409089.150219708
#Sta/Elev= 30
       0 2504.67    34.6 2484.89    93.1 2453.19   104.7 2445.81   110.5  2441.1
   115.1 2439.69   139.5  2435.5   156.9 2434.94   252.5 2434.25   264.2 2433.13
   295.1 2434.36   323.5 2433.27   356.9 2434.91   388.8 2433.53   408.7 2431.49
   417.1 2431.98   422.9 2433.44   432.1 2435.26   503.4 2434.05   667.1 2438.39
   690.3 2441.22   697.9  2444.5   704.6 2448.73   710.3 2450.17   738.9  2450.3
   757.3 2460.03   763.9 2462.29   780.1 2465.04   800.3 2467.22   850.6 2470.73
#Mann= 6 ,-1,0
       0      .1       0   388.8    .045       0   422.9      .1       0
     510     .07       0     600     .05       0     630     .06       0
Bank Sta=388.8,422.9
XS Rating Curve= 0 ,0
Exp/Cntr=0.3,0.1

Type RM Length L Ch R = 1 ,31023   ,218.8,222.3,225.5
XS GIS Cut Line= 3
 2230465.6604701409777.2731704352230953.44480959409485.543629775
2231049.11955142409363.205435305
#Sta/Elev= 30
       0 2492.34    26.2 2478.16    68.2 2457.82    86.8 2450.99   100.8 2447.25
   114.8 2444.54   127.3  2439.9   142.8 2439.63   152.1 2438.25   161.4 2435.66
   175.4 2435.44   191.5 2430.84   197.3 2430.03     234 2431.54   249.8 2430.44
   273.3 2431.35   299.4 2431.06   319.7 2429.06   324.5 2429.46   331.5 2431.27
   343.2 2431.53   366.5 2429.72   386.9 2431.52   483.1 2431.37   631.2 2435.63
   644.2 2437.08   657.2 2441.28   689.7 2440.19   702.7 2445.05   723.7 2449.96
#Mann= 6 ,-1,0
       0      .1       0     230     .07       0   299.4    .045       0
   331.5     .07       0     460     .05       0  578.37     .06       0
Bank Sta=299.4,331.5
XS Rating Curve= 0 ,0
Exp/Cntr(USF)=0,0
Exp/Cntr=0.3,0.1

Type RM Length L Ch R = 1 ,30801   ,323.5,324.2,322.9
XS GIS Cut Line= 4
2230589.74480703409948.4062674572230789.38097808 409833.15239551
2230829.51402278 409816.687556662231162.92700948409607.789913756
#Sta/Elev= 30
       0 2480.15    22.5 2467.11    35.1 2458.63    48.1 2451.79    62.8 2442.43
    77.3 2436.96   104.4 2433.59     133 2431.38   182.5 2429.23   206.5 2429.54
   222.5 2427.52   238.8  2428.6   244.9 2427.08   250.8 2426.78   255.2 2426.81
   263.3 2428.64   284.2 2429.51   303.1 2428.77   310.6 2429.43   340.8 2428.22
   399.8 2428.77   423.4 2428.15   571.5 2430.72   591.8 2431.62   603.4 2433.23
   612.1  2437.3     615 2437.67   641.1  2436.8   649.7  2441.8   667.3 2455.78
#Mann= 9 ,-1,0
       0      .1       0     200     .07       0   238.8    .045       0
   263.3     .07       0   313.9     .05       0   393.9     .07       0
   423.9     .05       0   573.9     .06       0   653.9      .1       0
Bank Sta=238.8,263.3
XS Rating Curve= 0 ,0
Exp/Cntr(USF)=0,0
Exp/Cntr=0.3,0.1

Type RM Length L Ch R = 1 ,30476   ,77.6,79.8,82.8
XS GIS Cut Line= 2
2230578.75637479410193.9032387712231322.31630005409901.870639728
#Sta/Elev= 30
       0 2489.14    31.6 2483.55    70.3 2472.78    97.3 2462.92     109 2458.15
   130.4 2448.99   143.3 2442.71   168.3 2440.04   208.4 2437.41   259.4 2431.19
   285.2 2429.76   323.8 2426.22   396.9 2426.69   430.5 2426.11   461.4 2426.34
   473.7 2425.76   486.1 2426.28   495.7 2424.84     500 2424.92   508.6 2426.31
   517.2 2425.29   534.4 2426.39     554 2425.75   624.9 2426.56     659 2427.47
   727.8 2430.46   763.8 2430.47   778.9 2431.99   788.5 2433.88   798.9 2434.26
#Mann= 11 ,-1,0
       0     .12       0      90     .06       0     120     .12       0
     200     .05       0     390     .07       0     410     .05       0
   486.1    .045       0   508.6     .05       0     510     .07       0
     660     .05       0     730     .06       0
Bank Sta=486.1,508.6
XS Rating Curve= 0 ,0
Exp/Cntr(USF)=0,0
Exp/Cntr=0.5,0.3

Type RM Length L Ch R = 1 ,30397   ,53.9,50.8,50.1
XS GIS Cut Line= 4
2230585.49558861410238.831330931 2230974.1235858410110.786268274
  2231196.517642410054.6261530732231344.78034613 409910.85625816
#Sta/Elev= 30
       0 2470.92    23.9 2466.78    61.8 2455.85    70.2 2454.03    87.1 2451.06
    99.7 2450.97   116.5 2448.58   120.7 2447.31   129.2 2443.29   133.3 2442.63
     190 2442.14   251.3 2438.34   301.8 2430.71   339.2 2429.08     365 2426.62
   386.1 2426.24     436 2426.81   481.1 2425.21   493.8 2424.36   514.4 2424.41
   525.7 2425.35   535.1 2425.93   584.6 2424.89   710.5 2426.36   755.3 2429.74
   788.5 2431.14   803.4 2430.09   816.4 2430.62   827.5 2433.55   845.1 2434.16
#Mann= 8 ,-1,0
       0     .12       0      80     .06       0     190     .05       0
   481.1    .045       0   525.7     .05       0  648.55     .07       0
  718.55     .05       0  788.55     .06       0
#XS Ineff= 2 , 0
          474.01  2426.9  529.93            2426
Permanent Ineff=
       F       F
Bank Sta=481.1,525.7
XS Rating Curve= 0 ,0
Exp/Cntr(USF)=0,0
Exp/Cntr=0.5,0.3

Type RM Length L Ch R = 1 ,30346   ,199.4,193.5,199.2
XS GIS Cut Line= 4
2230588.08574656410293.6872433272231038.50567098410146.751381568
2231227.96730651410097.3078406262231413.04935853409928.847536386
#Sta/Elev= 30
       0 2447.56    29.5 2447.41      80 2444.06   156.4 2441.29   172.6 2441.22
   193.6 2442.34   223.1 2441.95     261 2438.99   286.2 2435.59   374.6 2429.78
   416.6 2427.49     492 2426.91   511.7 2424.77   525.1 2423.12   533.4 2423.51
   537.5 2424.89   607.8 2424.21   624.3 2425.14   661.5 2424.26   771.8 2426.79
   794.3 2426.18   832.1 2426.74   848.1  2427.2   853.8 2429.14   859.9 2432.42
   880.8 2434.16   886.2 2433.68   899.2 2428.66   913.3 2428.86   919.9 2429.86
#Mann= 10 ,-1,0
       0     .12       0      80      .1       0     150     .06       0
     180     .05       0   511.7    .045       0   537.5     .05       0
  699.59      .1       0  739.59     .05       0  839.59     .06       0
  889.59     .07       0
#XS Ineff= 2 , 0
          510.79  2426.4  538.25            2426
Permanent Ineff=
       F       F
Bank Sta=511.7,537.5
XS Rating Curve= 0 ,0
Exp/Cntr=0.5,0.3

Type RM Length L Ch R = 1 ,30152   ,200,201.2,194.6
XS GIS Cut Line= 3
2230632.67008538410380.3548212372231090.93662542410254.556163188
 2231560.4351885410041.147725425
#Sta/Elev= 30
       0 2448.13    11.9 2446.69    57.3 2444.57    74.2 2445.63   129.1 2445.87
   190.3  2439.4   329.3 2431.79   412.3 2428.17   476.6 2424.26   534.6  2424.2
   546.2  2423.5     598 2423.35   613.9 2422.26   630.4  2422.5   640.3 2421.71
   662.2 2422.46   673.5 2423.46   696.3 2422.66   721.9 2423.79   740.2 2423.52
   749.1 2424.34   766.6 2428.08   784.1 2429.36   858.8 2431.57     885 2433.84
   894.1 2433.87   903.1 2431.82   924.8 2433.62   942.2 2436.89   990.9 2452.35
#Mann= 8 ,-1,0
       0     .12       0      30      .1       0     240     .05       0
   630.4    .045       0   662.2      .1       0  765.22     .06       0
  965.22     .07       0  975.22      .1       0
Bank Sta=630.4,662.2
XS Rating Curve= 0 ,0
Exp/Cntr(USF)=0,0
Exp/Cntr=0.3,0.1

Type RM Length L Ch R = 1 ,29951   ,116.4,117.5,111.2
XS GIS Cut Line= 3
2230915.93482126410370.0028205492231185.70622445410435.877232956
2231591.93176763410191.200844016
#Sta/Elev= 30
       0 2433.99    70.2 2430.28   197.9 2425.35   226.7 2424.99   267.6 2423.12
   299.3 2423.31   322.6 2421.34   344.9 2422.37   369.3 2422.38   397.3 2419.45
   430.2 2420.55   439.3 2421.55   447.6 2420.72   459.2 2419.15     472 2418.94
   485.5 2420.79   507.8 2420.84   523.3 2419.84   546.5 2420.59   565.4 2426.04
   619.5 2426.71   674.9 2429.16   678.3 2429.92   686.8 2435.09   691.5 2436.34
     704 2436.22   714.8 2435.23   718.6 2435.77   732.6 2444.75   751.9  2452.6
#Mann= 7 ,-1,0
       0      .1       0      40     .05       0   357.7      .1       0
   447.6    .045       0   485.5      .1       0   647.7     .07       0
   697.7      .1       0
#XS Ineff= 2 , 0
          300.52 2427.79
Permanent Ineff=
       F       F
Bank Sta=447.6,485.5
XS Rating Curve= 0 ,0
Exp/Cntr(USF)=0,0
Exp/Cntr=0.3,0.1

Type RM Length L Ch R = 1 ,29834   ,497.3,515,510.4
XS GIS Cut Line= 3
2230947.80264052 410668.990807442231062.06004978410627.109405225
2231628.50771745410273.243718955
#Sta/Elev= 30
       0 2492.03    34.5 2474.36   106.1 2435.54   128.9 2427.53   144.9 2424.64
   176.1 2422.42   312.8 2421.28   336.7 2420.21   409.1 2421.06   420.7  2418.9
     426 2418.71   442.4 2419.96     473 2419.17   501.5  2420.9   562.8 2419.44
   580.4 2418.04   586.4 2418.18     592 2419.52     601 2420.82     610 2423.83
   615.2 2424.47     684 2426.18   719.7 2429.22   727.9 2432.24   737.3 2437.92
   746.7 2438.35   760.9 2437.58   765.6 2438.72   783.6 2452.26   789.6 2455.45
#Mann= 6 ,-1,0
       0      .1       0  231.69     .05       0  351.69      .1       0
   562.8    .045       0     592      .1       0  691.69     .06       0
#XS Ineff= 2 , 0
          212.98 2431.95
Permanent Ineff=
       F       F
Bank Sta=562.8,592
XS Rating Curve= 0 ,0
Exp/Cntr=0.3,0.1

Type RM Length L Ch R = 1 ,29319   ,317.6,311.9,307.7
XS GIS Cut Line= 3
     2230919.912      410846.929     2231385.939      410868.659
     2231840.377      410797.216
#Sta/Elev= 30
       0 2537.04    52.3 2513.89    76.3 2501.22    96.4 2489.33   172.5 2451.09
   201.4 2442.16   216.7 2436.23   228.5 2430.63   248.5 2424.69   264.6 2422.11
   372.7  2416.2   404.7 2416.86   416.7 2415.01   436.7 2416.48   451.5 2416.58
   456.8 2415.61   464.8 2413.56   493.1 2414.29   498.7 2415.42   505.2 2417.22
   509.3 2417.34   557.9 2415.45     566 2418.25   574.1 2423.14   578.1 2424.45
   597.5  2427.8   675.3 2431.46   767.7 2437.29   849.4  2440.5   926.6 2444.57
#Mann= 5 ,-1,0
       0      .1       0   456.8    .045       0   498.7      .1       0
  656.53     .05       0  826.53     .06       0
Bank Sta=456.8,498.7
XS Rating Curve= 0 ,0
Exp/Cntr=0.3,0.1

Type RM Length L Ch R = 1 ,29007   ,227.8,226.1,218.4
XS GIS Cut Line= 5
2231153.51654253411243.7838880022231381.15615994411142.620094433
  2231536.929508411110.0666173092231596.94384561411084.870156131
2231861.17363757410863.150519972
#Sta/Elev= 30
       0 2482.35    24.8 2486.24    42.3 2487.66    51.1 2487.65    59.8 2486.46
    68.6 2483.85    81.7 2478.52    90.5 2473.68   113.1 2458.68   155.5 2427.75
   176.7 2415.35   182.4 2414.64   191.9 2415.08   204.3  2412.5   234.9 2414.01
     248 2412.56   272.6 2410.88   276.7    2411   284.9 2413.05   301.2 2412.59
   325.7 2413.81   407.5 2414.05   429.7 2414.77   442.6  2416.1   459.5 2420.93
   468.2 2422.67   492.4 2425.07   702.5 2436.72   777.8 2439.59   818.3 2442.07
#Mann= 4 ,-1,0
       0      .1       0     248    .045       0   284.9      .1       0
  418.24     .05       0
Bank Sta=248,284.9
XS Rating Curve= 0 ,0
Exp/Cntr(USF)=0,0
Exp/Cntr=0.3,0.1

Type RM Length L Ch R = 1 ,28781   ,155.3,154.3,154.4
XS GIS Cut Line= 2
2231313.81321267 411408.427630472232036.66801005 411001.79552489
#Sta/Elev= 30
       0 2499.85    33.5 2476.36      67 2451.27    94.5 2426.98   108.3 2411.55
   112.8 2409.32   131.2 2409.29   137.2 2411.12     145 2412.03   172.5 2410.86
   190.9 2412.41   259.5 2412.12   312.5 2413.06     333 2414.32   351.5 2418.54
   365.6 2420.01   420.4 2421.88   485.8 2425.65   511.7 2425.84   562.6 2424.22
   594.8  2426.3   626.9 2426.97   672.8 2430.11   732.5 2436.32   746.2 2440.77
   769.1 2439.64   773.7 2440.36   778.3 2443.45   796.7 2459.61   829.4 2472.87
#Mann= 6 ,-1,0
       0      .1       0   108.3    .045       0   137.2      .1       0
     160     .05       0     720     .06       0  829.38      .1       0
Bank Sta=108.3,137.2
XS Rating Curve= 0 ,0
Exp/Cntr=0.3,0.1

Type RM Length L Ch R = 1 ,28626   ,351.3,353.5,351.9
XS GIS Cut Line= 3
2231307.24284998411592.9772629752231762.90726514 411322.54228487
2232016.67159391411197.512414856
#Sta/Elev= 30
       0 2547.68    47.6 2517.29    67.7 2504.99   114.4 2473.19   126.7 2463.95
   155.2 2436.13   168.5 2425.35   179.9 2413.93   182.5  2411.8   187.7 2409.87
   196.4 2408.78   216.5 2409.46   242.8 2408.84   258.2 2410.39   273.9 2410.61
   289.5 2411.68   298.8 2411.23   340.6 2411.73   401.1 2413.55   433.7 2413.94
   461.6 2413.45   484.8 2415.77   553.6 2417.56   582.6 2420.61   594.6 2421.34
   621.5 2422.39   668.7 2423.05   797.7 2427.27   806.7 2429.57   812.8 2432.74
#Mann= 7 ,-1,0
       0      .1       0   187.7    .045       0   216.5      .1       0
     320     .05       0  619.87     .06       0  729.87     .05       0
  739.87     .06       0
#XS Ineff= 2 , 0
                          371.24         2422.01
Permanent Ineff=
       F       F
Bank Sta=187.7,216.5
XS Rating Curve= 0 ,0
Exp/Cntr(USF)=0,0
Exp/Cntr=0.3,0.1

Type RM Length L Ch R = 1 ,28273   ,443.2,445.9,443.4
XS GIS Cut Line= 2
2231456.38893162411902.6325077952232239.83645802411455.325201107
#Sta/Elev= 30
       0 2533.36    13.6 2524.55    67.5 2492.29    91.9 2474.88   115.3 2455.05
   128.7 2440.66   140.1 2430.77   151.8 2418.38   159.2 2411.85   165.1 2407.65
   172.3 2406.08   188.6 2405.97   194.4 2406.77     212 2406.66   225.4 2405.43
   234.7 2405.92   243.9 2409.01   248.5 2409.68   349.8 2408.22   474.2  2408.7
   519.9 2410.09   640.3 2410.94   745.9 2415.71   787.4 2419.78   801.2 2425.06
   805.8 2426.19   828.8 2425.64   833.4 2426.28   842.4 2432.44   902.1 2457.08
#Mann= 5 ,-1,0
       0      .1       0   165.1    .045       0   194.4      .1       0
     330     .05       0     790     .06       0
#XS Ineff= 2 , 0
                          454.69         2424.49
Permanent Ineff=
       F       F
Bank Sta=165.1,194.4
XS Rating Curve= 0 ,0
Exp/Cntr=0.3,0.1

Type RM Length L Ch R = 1 ,27827   ,315.7,325.5,311.4
XS GIS Cut Line= 3
 2231676.0738018412249.8083936682232165.45116741412013.533617198
2232401.17723982411864.994946607
#Sta/Elev= 30
       0  2456.3    17.9 2448.92    45.5  2436.2    57.9 2426.51    75.6 2407.11
    78.4 2404.66    84.4 2403.15   108.4 2404.41   128.9  2402.7   139.4 2403.29
   146.7 2402.54     162 2404.21   195.3 2402.87   204.4  2403.7   225.2    2403
   244.4 2405.55   262.2 2404.96     342 2405.75   395.4 2405.34   416.9  2406.1
     431 2404.89   713.9 2409.08   725.5 2411.27   735.8 2417.98   740.5 2419.76
   764.1 2419.16   768.9 2420.05   792.5 2433.96   811.4 2447.03   822.1 2450.86
#Mann= 8 ,-1,0
       0      .1       0    78.4    .045       0   108.4      .1       0
     190     .07       0     410     .05       0     530      .1       0
  633.43     .06       0  743.43      .1       0
#XS Ineff= 2 , 0
                          376.34          2413.7
Permanent Ineff=
       F       F
Bank Sta=78.4,108.4
XS Rating Curve= 0 ,0
Exp/Cntr=0.3,0.1

Type RM Length L Ch R = 1 ,27501   ,153.3,151.4,144.3
XS GIS Cut Line= 3
2231690.64124671412497.0364911512232077.56495967412301.516529812
2232436.70425708412081.299310199
#Sta/Elev= 30
       0 2502.23    33.1 2484.99      60 2473.29   104.8 2452.69   123.1 2442.33
   150.5 2427.89   167.5 2414.31     172  2411.5   188.6 2404.14   197.5 2401.36
   212.4 2400.23   221.4 2400.91   257.1 2401.44     266 2399.72     269  2399.7
   283.9 2399.91     293 2401.13   301.7 2401.25     311 2403.29   355.8  2402.3
   409.6 2404.39     456 2403.76   587.2 2404.03   718.1 2406.78   755.6 2408.25
   832.1 2408.98   835.4 2409.06     840 2410.18   847.4 2413.57   854.8 2414.52
#Mann= 6 ,-1,0
       0      .1       0   257.1    .045       0   301.7      .1       0
     410     .07       0  733.52      .1       0  853.52     .06       0
#XS Ineff= 2 , 0
                          410.85         2419.29
Permanent Ineff=
       F       F
Bank Sta=257.1,301.7
XS Rating Curve= 0 ,0
Exp/Cntr(USF)=0,0
Exp/Cntr=0.3,0.1

Type RM Length L Ch R = 1 ,27350   ,64.5,62.2,53.9
XS GIS Cut Line= 2
2231785.32073204412668.5463738582232479.51164787412151.219385631
#Sta/Elev= 30
       0 2485.35    24.5 2471.75    58.4 2449.21    67.3 2444.02    78.8 2438.33
    92.7 2433.72    99.4 2430.49   132.8 2410.58   143.2 2405.31   153.2 2403.03
   168.2 2401.33   213.2 2400.63     243 2401.29   253.3 2399.23   258.8 2398.12
   267.4  2397.9   277.9 2398.91   287.9 2398.21     296 2399.09   317.8 2401.17
   360.4 2400.72     396 2402.94   514.4  2403.3   532.3 2402.75   746.9 2407.38
   807.7 2406.82     842 2407.68   850.5 2409.61   856.6 2412.61   865.8 2414.38
#Mann= 7 ,-1,0
       0      .1       0     200     .08       0   253.3    .045       0
     296      .1       0     560     .07       0     690      .1       0
     810     .06       0
#XS Ineff= 2 , 0
                          498.44         2412.69
Permanent Ineff=
       F       F
Bank Sta=253.3,296
XS Rating Curve= 0 ,0
Exp/Cntr(USF)=0,0
Exp/Cntr=0.5,0.3

Type RM Length L Ch R = 1 ,27288   ,41.2,41.8,42.3
XS GIS Cut Line= 4
2231800.05939267412705.3930254412231932.70733837412675.915704175
 2232112.5189981412472.522187436 2232510.4628352412214.595626354
#Sta/Elev= 30
       0 2483.38      37 2460.32    53.4 2449.51    65.7 2440.17    94.4 2421.98
   110.8 2414.89   135.3  2401.5   140.3 2400.66   162.9 2400.42   228.1 2399.96
   267.7 2400.81     289 2400.66   294.4 2399.74   299.7 2397.99   313.1 2397.83
   328.3 2399.62   357.7 2400.94   418.2  2402.4   442.9 2402.09   521.4 2402.45
   557.4 2403.28   678.3 2405.58   754.9 2406.91   788.4 2406.55   807.4 2405.71
   821.7 2406.86   850.3 2407.07   857.8 2408.37   869.3  2412.9   881.6 2414.54
#Mann= 11 ,-1,0
       0      .1       0   162.9     .06       0   228.1     .08       0
   294.4    .045       0   328.3     .08       0   357.7      .1       0
   442.9     .07       0   521.4      .1       0   557.4     .07       0
   678.3      .1       0   788.4     .06       0
#XS Ineff= 3 ,-1
     100     278    2400     343   418.2    2400   418.2     550    2405
Permanent Ineff=
       F       F       F
Bank Sta=294.4,328.3
XS Rating Curve= 0 ,0
Exp/Cntr(USF)=0,0
Exp/Cntr=0.5,0.3

Type RM Length L Ch R = 1 ,27246   ,67.4,69.7,72
XS GIS Cut Line= 4
2231819.40023982412743.068053393 2231950.1185629412709.853525789
 2232140.5224533412507.8949729562232556.38606154412223.568267873
#Sta/Elev= 30
       0 2476.98    33.8 2455.83    77.9 2425.17     104 2410.74   128.7 2401.24
   137.9 2400.11   184.9  2399.5   207.8 2400.35   235.8 2399.35   295.2 2400.37
   311.7 2399.69   324.5 2397.85     342 2399.47     400 2400.94   426.6 2403.12
   437.2 2401.79   513.8 2401.88   567.1 2403.59   688.2 2405.65   750.9 2406.34
   794.8 2405.52     817 2406.95   837.2 2407.33   843.3 2406.74   851.6 2408.26
   857.8 2411.71   862.6 2413.03   891.7    2415   906.2 2425.49   916.2 2431.62
#Mann= 11 ,-1,0
       0      .1       0  134.87     .06       0  264.87      .1       0
  274.87     .08       0   311.7    .045       0     342     .08       0
  404.87      .1       0  412.43     .07       0  652.43      .1       0
  772.43     .06       0  892.43      .1       0
#XS Ineff= 2 , 0
           309.2    2400  344.96          2400.3
Permanent Ineff=
       F       F
Bank Sta=311.7,342
XS Rating Curve= 0 ,0
Exp/Cntr=0.5,0.3

Type RM Length L Ch R = 1 ,27176   ,434,445.8,439.8
XS GIS Cut Line= 4
2231832.17905759412787.7370235062231939.34627039412779.677301747
2232263.82344916412505.2689105762232526.86786337412287.007564939
#Sta/Elev= 30
       0 2474.41    40.1 2448.42    60.2 2436.66    72.2 2430.78   107.5 2415.71
   129.5 2402.04   132.5 2401.16     140 2400.04   169.4 2399.45   202.9 2400.82
   222.8 2400.32   231.9 2399.09   244.8 2398.76   260.3 2399.56   328.1 2400.07
   351.7 2398.46   365.2 2397.28   376.6 2397.36   382.22398.688   390.1 2400.72
   396.3 2401.19   501.6 2401.06   761.6 2405.68   795.7 2405.77   819.6  2404.9
   836.7  2406.3   849.9 2406.35   856.6  2407.9   865.5 2412.25   874.2  2413.4
#Mann= 8 ,-1,0
       0      .1       0  217.47     .06       0  237.47      .1       0
   351.7    .045       0   382.2      .1       0  497.47     .07       0
  622.42      .1       0  752.42     .06       0
Bank Sta=351.7,382.2
XS Rating Curve= 0 ,0
Exp/Cntr(USF)=0,0
Exp/Cntr=0.3,0.1

Type RM Length L Ch R = 1 ,26731   ,247.1,246.8,245.4
XS GIS Cut Line= 5
2231984.48438328412953.8106549062232094.02979852412924.093248813
2232344.08953855412805.7522195822232602.29978559412687.771122257
2232622.57263078412644.580708917
#Sta/Elev= 30
       0 2429.93    41.1 2422.16      66 2416.81      95 2412.35    99.1 2411.15
   111.6  2403.9   128.7 2396.72   142.4  2394.7   153.3 2394.54   157.7 2394.88
   163.72396.706   167.1 2397.17   182.3 2396.93   222.1 2397.89   401.2 2397.69
   429.9 2398.44   482.6 2398.93   491.4 2399.47   511.4  2398.3   526.5 2399.72
   566.2 2399.62   623.1 2401.24   654.1  2401.4   659.3 2401.92   662.9 2402.99
   671.7 2407.83     674  2408.8   678.5 2409.78   694.6 2410.58   721.8 2410.73
#Mann= 3 ,-1,0
       0     .12       0   128.7    .045       0   163.7      .1       0
#XS Ineff= 2 , 0
                          489.11         2403.72
Permanent Ineff=
       F       F
Bank Sta=128.7,163.7
XS Rating Curve= 0 ,0
Exp/Cntr=0.3,0.1

Type RM Length L Ch R = 1 ,26484   ,185.2,197.6,204.2
XS GIS Cut Line= 3
2231941.73003917413171.0658315582232136.22094808413179.298250982
2232670.29915826412903.512200251
#Sta/Elev= 30
       0 2448.88    10.5  2443.5    42.5 2430.69    62.5 2424.45   106.5 2412.03
   118.6 2409.02   162.6 2401.14   196.2 2397.04   217.1 2395.62   234.2  2395.5
   249.6 2394.68   280.1 2395.16   289.2 2394.81   297.1 2394.01     309 2393.68
   332.8 2394.02   338.6 2394.94   343.2 2396.16   347.5 2396.29   374.3 2395.28
   415.9  2395.3   433.2 2394.38   473.7 2395.17   527.7 2395.02   545.8 2395.91
   626.5 2397.36   766.2 2402.78   774.7 2404.81     784 2408.74   795.7 2409.47
#Mann= 5 ,-1,0
       0     .12       0  194.67      .1       0   289.2    .045       0
   338.6      .1       0  754.67     .06       0
Bank Sta=289.2,338.6
XS Rating Curve= 0 ,0
Exp/Cntr(USF)=0,0
Exp/Cntr=0.3,0.1

Type RM Length L Ch R = 1 ,26286   ,109,102.4,101.7
XS GIS Cut Line= 3
2231985.72993665 413351.492196382232539.05669502413258.501937557
2232765.66424977413175.507017193
#Sta/Elev= 30
       0 2449.07    18.7 2440.88      39 2434.88   102.5 2413.74   144.4 2402.41
   160.7    2399   209.8 2394.63   245.8 2394.86   266.1 2391.91   278.3 2393.75
   290.5 2393.03   302.6  2391.5   310.7  2391.6   318.9 2393.41   359.4 2394.65
     400 2394.56   456.8 2392.84   533.8 2392.18   583.6 2393.38   617.7  2393.2
     639 2394.57     656 2396.91   698.6 2397.91   732.7 2402.13   745.5  2406.5
     754 2410.97   775.3 2410.27   779.5 2410.87   793.7 2422.13   802.4 2427.49
#Mann= 6 ,-1,0
       0      .1       0      60     .12       0     260      .1       0
   290.5    .045       0   318.9      .1       0  731.09     .06       0
Bank Sta=290.5,318.9
XS Rating Curve= 0 ,0
Exp/Cntr=0.3,0.1

Type RM Length L Ch R = 1 ,26184   ,406.8,379.2,364.1
XS GIS Cut Line= 3
2232011.70560428413444.793777433  2232616.788432413351.150006475
2232791.72734478413264.709602515
#Sta/Elev= 30
       0 2451.71    49.1 2430.05     130 2400.83   162.4 2395.89   182.3 2394.15
     215  2393.1   234.9  2393.7   240.5 2392.09   243.3 2390.94     259 2390.16
   275.7 2391.39   287.9 2390.65   298.32392.423   308.1 2393.76   385.6 2391.08
   413.3 2392.43   494.4  2392.5   518.6 2390.73   546.9 2392.59   578.4 2391.99
   587.4 2393.17   603.6 2398.66   611.7 2399.89     673 2399.88   718.7 2401.51
   745.5 2404.48   758.8 2410.17   763.3 2410.91   789.5 2408.46   807.4 2418.74
#Mann= 10 ,-1,0
       0      .1       0      30     .12       0     230      .1       0
   240.5    .045       0   298.3      .1       0     330     .05       0
     430      .1       0  632.29     .07       0  732.29      .1       0
  742.29     .06       0
Bank Sta=240.5,298.3
XS Rating Curve= 0 ,0
Exp/Cntr(USF)=0,0
Exp/Cntr=0.3,0.1

Type RM Length L Ch R = 1 ,25804   ,69.2,86.9,103.6
XS GIS Cut Line= 4
2232048.24478782413666.3734059142232473.96630613413568.958820577
2232560.59247723 413449.768170932232827.36223469413281.747439711
#Sta/Elev= 30
       0 2453.38    20.4 2441.74    36.9 2430.78    73.8 2410.92   110.7 2398.22
   135.3 2394.33   168.2 2392.37     242 2392.42   261.4 2390.67     320  2391.8
   356.9 2391.54   373.3 2389.66   393.9 2392.43   490.8  2390.9     5012388.985
   510.6 2387.32   525.5 2387.22   535.5 2388.71   587.1 2388.77   598.7 2395.04
   611.9 2398.12   659.2  2400.4   712.8  2400.3   796.3 2402.63   824.7 2405.66
   833.6 2409.54   838.8 2410.23   862.6 2407.42   870.4 2411.49   899.3 2432.79
#Mann= 10 ,-1,0
       0      .1       0      90     .06       0     320     .05       0
     400      .1       0     501    .045       0   535.5      .1       0
  536.72     .07       0  664.07     .06       0  684.07     .07       0
  784.07     .06       0
Bank Sta=501,535.5
XS Rating Curve= 0 ,0
Exp/Cntr(USF)=0,0
Exp/Cntr=0.5,0.3

Type RM Length L Ch R = 1 ,25718   ,60.7,60.1,57.7
XS GIS Cut Line= 4
2232056.53028357413681.1651428722232623.96871795413545.569465046
 2232762.5121279413457.137501246 2232850.9440917413303.855430661
#Sta/Elev= 30
       0  2450.6    61.3 2414.49    81.9 2403.98    90.1 2402.14   110.7 2396.32
   147.7 2392.54   242.3 2392.38   271.9 2390.27   332.8 2391.23   349.2 2389.76
   371.5 2392.69   390.3 2391.97   497.3    2391   512.9 2390.04   521.9 2387.23
   542.5 2386.61   550.7 2387.31   557.4 2390.48   563.1 2392.03   595.4  2393.9
   621.6  2396.3   650.1 2396.32   695.7 2399.11   799.1 2401.56   841.4 2404.37
   872.4 2408.43   895.5 2406.06   900.1  2407.8   918.8 2424.77   924.7  2427.7
#Mann= 8 ,-1,0
       0      .1       0    90.1     .06       0   371.5     .05       0
   390.3      .1       0   497.3     .07       0   512.9    .045       0
   557.4     .07       0   595.4     .06       0
#XS Ineff= 2 , 0
           504.9  2392.6  559.43          2393.2
Permanent Ineff=
       F       F
Bank Sta=512.9,557.4
XS Rating Curve= 0 ,0
Exp/Cntr(USF)=0,0
Exp/Cntr=0.5,0.3

Type RM Length L Ch R = 1 ,25657   ,100.2,100.6,103.4
XS GIS Cut Line= 3
2232100.75724018413758.2263411772232646.21613405413597.573052735
2232923.40305242413428.026164677
#Sta/Elev= 30
       0 2433.88    11.9 2427.44    24.4 2418.81    28.6 2416.55    45.3 2409.72
    55.1 2404.43    78.6 2393.69    99.5 2392.22   178.7 2391.27   287.2 2391.72
   393.4 2391.11   444.9 2390.07   462.3 2390.36   474.8 2392.58   478.9 2392.36
   482.3 2389.92   487.3  2387.5   495.6  2385.8   512.3 2386.53     529 2389.72
   533.1 2391.14   541.5 2392.41   683.5 2396.18   730.3 2398.78   785.6 2400.81
   814.7 2402.87     838  2403.5     871 2406.07   880.4 2406.32   893.6 2405.22
#Mann= 11 ,-1,0
       0      .1       0      40     .06       0     140     .05       0
     230     .06       0   482.3    .045       0     529     .06       0
     550     .05       0  578.63     .06       0  668.63     .05       0
  768.63     .06       0  893.55     .05       0
#XS Ineff= 2 , 0
          480.97 2391.41  530.82         2391.41
Permanent Ineff=
       F       F
Bank Sta=482.3,529
XS Rating Curve= 0 ,0
Exp/Cntr=0.5,0.3

Type RM Length L Ch R = 1 ,25557   ,114.3,112.3,109.3
XS GIS Cut Line= 2
2232094.85080122413856.5552044072232933.48059125413622.210500339
#Sta/Elev= 30
       0 2443.53     9.7 2438.88    22.1 2431.62    30.4  2429.4      72 2406.22
    84.4 2400.76    92.7 2395.07    96.9 2393.98   105.2 2393.79   113.5 2391.88
   238.1 2390.08   379.3 2389.54   425.8 2390.24   487.3 2388.84   499.8 2389.69
     507 2388.67   512.2    2387   520.5 2386.14   529.7 2386.36   537.1 2388.69
   541.3  2389.6   566.2 2390.42   603.6 2390.26   703.3 2398.74     778  2402.3
   812.1 2409.61     832 2415.77   844.3 2421.72   852.8 2423.55   870.8 2429.29
#Mann= 6 ,-1,0
       0      .1       0      50     .06       0     240     .05       0
     507    .045       0   537.1     .05       0     860      .1       0
#XS Ineff= 2 , 0
             189 2398.59
Permanent Ineff=
       F       F
Bank Sta=507,537.1
XS Rating Curve= 0 ,0
Exp/Cntr(USF)=0,0
Exp/Cntr=0.3,0.1

Type RM Length L Ch R = 1 ,25445   ,129.4,125.6,120.1
XS GIS Cut Line= 4
2232106.37842766413903.7511603662232372.90300654413929.477471068
2232766.00103407413764.8290825722232913.15553129413674.272468899
#Sta/Elev= 30
       0    2442     9.8 2436.72    25.9 2430.51    66.1 2411.56    74.1 2407.37
    86.2 2399.08    94.2 2394.64   110.3 2393.91   118.3 2390.95   164.2 2390.07
   226.8 2390.62   336.4 2388.66   427.4 2388.89   470.8 2388.14   522.8 2389.51
     527 2388.51   531.5 2386.22   548.6 2385.73   558.4 2388.34   561.9 2389.23
   574.9 2388.36   600.9  2389.1   652.9 2388.24   674.6 2390.09   700.9 2394.23
   729.4 2397.59   799.9 2400.45   842.1 2408.48   856.2 2416.34   866.7 2418.95
#Mann= 7 ,-1,0
       0      .1       0     130     .06       0     230     .05       0
     527    .045       0   558.4     .05       0  657.76      .1       0
  833.95     .05       0
#XS Ineff= 2 , 0
          289.62 2395.23
Permanent Ineff=
       F       F
Bank Sta=527,558.4
XS Rating Curve= 0 ,0
Exp/Cntr(USF)=0,0
Exp/Cntr=0.3,0.1

Type RM Length L Ch R = 1 ,25319   ,206.2,207.9,211.2
XS GIS Cut Line= 3
2232138.29393846 414128.845428962232436.45723349414107.258463346
2232953.73144706413744.880035293
#Sta/Elev= 30
       0 2438.23     9.9 2432.65    21.9 2428.08      54 2412.31    94.1 2394.53
    98.1 2393.41   106.2 2393.31   114.2  2390.6   162.3  2389.5   397.9 2387.61
   464.7 2387.78   498.8 2386.35   578.8 2389.09   584.6 2387.98   588.4 2386.38
   593.2 2385.93   613.3 2386.06   620.9 2387.76   639.1 2388.17   658.1 2387.15
   669.8 2388.05   718.6 2388.34   736.8 2390.61   762.7 2390.38   837.3 2393.42
   850.5 2394.98   868.9 2398.39   879.8  2405.1   897.6 2410.36   930.5 2423.68
#Mann= 6 ,-1,0
       0      .1       0     100     .06       0     200     .05       0
   584.6    .045       0   620.9     .05       0  778.94      .1       0
#XS Ineff= 2 , 0
           200.4 2394.98
Permanent Ineff=
       F       F
Bank Sta=584.6,620.9
XS Rating Curve= 0 ,0
Exp/Cntr=0.3,0.1

Type RM Length L Ch R = 1 ,25111   ,119.7,119.3,123.3
XS GIS Cut Line= 3
2232139.30810536414144.5494285412232724.83893695414135.287956688
2233044.87424209413980.930092473
#Sta/Elev= 30
       0 2438.08    32.9 2422.18    84.9  2398.3    92.9 2394.11    96.9 2393.39
   108.9 2393.22   112.9 2391.44   116.9  2390.5   136.9 2389.71   168.9 2389.27
   312.9 2388.76   432.9 2386.67   476.8 2384.91   508.9 2385.35   524.9 2385.06
   551.6 2385.96   568.9 2385.78   589.7 2386.26   629.3 2385.34   664.8 2385.83
     687 2385.67   691.2 2386.23   697.5 2390.61   700.3 2392.12   704.8  2392.5
   721.5 2393.07   780.3 2397.61   841.3 2399.15   874.3 2400.77   940.9 2405.42
#Mann= 9 ,-1,0
       0      .1       0     100     .06       0     200     .05       0
     490     .07       0   595.6      .1       0   664.8    .045       0
   691.2      .1       0   695.6     .05       0   705.6      .1       0
Bank Sta=664.8,691.2
XS Rating Curve= 0 ,0
Exp/Cntr(USF)=0,0
Exp/Cntr=0.3,0.1

Type RM Length L Ch R = 1 ,24992   ,340.3,350.3,352.5
XS GIS Cut Line= 4
2232138.27905293414262.8904577732232529.31897561414314.343079178
2232874.05153902414199.089207231 2233023.2641411414265.977615057
#Sta/Elev= 30
       0 2440.57    18.1 2431.96    34.2 2422.94    42.3 2421.21    54.4 2414.51
    98.7 2394.26   114.9 2392.73   122.9 2389.88   195.6 2388.31   388.8 2387.66
   438.7  2386.3   469.1 2383.56   481.8  2384.4   494.4  2383.1   536.5 2385.09
   606.2 2385.85   637.9 2385.53   654.7  2383.2   663.1 2384.16   684.2 2383.41
   692.7 2384.25   713.7 2383.15   724.3 2384.46   730.6 2388.07     769 2391.77
   782.6 2394.61   799.7 2400.29   839.1 2417.13   869.8  2427.9   921.4 2440.83
#Mann= 8 ,-1,0
       0      .1       0     100     .06       0     200     .05       0
  504.41     .07       0  604.41      .1       0   692.7    .045       0
   724.3      .1       0   817.9     .12       0
Bank Sta=692.7,724.3
XS Rating Curve= 0 ,0
Exp/Cntr(USF)=0,0
Exp/Cntr=0.3,0.1

Type RM Length L Ch R = 1 ,24641   ,286.4,292,296.1
XS GIS Cut Line= 4
2232098.35587469414484.2058488332232565.90327483414562.484842296
2232926.53321286414539.7055609322233087.34793647414478.609354069
#Sta/Elev= 30
       0 2450.72    47.6 2426.38   119.5 2391.56   123.5 2390.68   139.7 2389.67
   147.8 2387.94   165.7 2387.02   204.6 2386.87   216.8 2386.15   245.2 2385.82
   549.1 2385.62   612.6 2383.22   636.7 2383.06   648.7 2383.52   660.7 2382.91
   700.8  2383.5   718.7 2382.95   732.8 2381.56   741.3 2381.42   760.9 2380.04
   776.9  2380.6     779 2381.66   800.2 2394.32     825 2406.57   871.4 2434.51
   888.2 2442.28   898.8 2444.43   918.5 2447.26   944.3 2449.58  1007.4 2456.92
#Mann= 8 ,-1,0
       0      .1       0     140     .07       0     240     .05       0
  634.06      .1       0  734.06     .07       0   741.3    .045       0
     779     .07       0  834.06      .1       0
#XS Ineff= 2 , 0
          481.93 2396.48
Permanent Ineff=
       F       F
Bank Sta=741.3,779
XS Rating Curve= 0 ,0
Exp/Cntr=0.3,0.1

Type RM Length L Ch R = 1 ,24349   ,300.2,311.5,314.3
XS GIS Cut Line= 3
2232061.09421017414731.4258617592232863.51454285414838.177190784
2233203.07301479414740.452214512
#Sta/Elev= 30
       0 2451.63    39.4 2432.79    63.6 2422.21     104 2406.16   116.1 2402.22
   148.4 2388.55   152.4    2388   164.5 2387.82   176.6 2385.85   237.2 2383.81
   595.5 2382.75   656.8 2380.63   693.1 2381.12   721.4  2380.9   723.32380.223
   729.5 2378.55   737.5 2378.47   753.7 2379.93   781.9 2379.67     794 2381.18
   818.5 2391.68   835.2 2397.26   851.8 2405.18   885.4 2418.65   905.9 2425.13
     935  2431.9  1022.5 2443.39  1068.2 2448.35  1124.3 2456.85  1162.8 2460.41
#Mann= 7 ,-1,0
       0      .1       0      80     .06       0     280     .05       0
   723.3    .045       0   753.7     .05       0     770      .1       0
 1039.49     .12       0
#XS Ineff= 2 , 0
           601.1 2399.38
Permanent Ineff=
       F       F
Bank Sta=723.3,753.7
XS Rating Curve= 0 ,0
Exp/Cntr=0.3,0.1

Type RM Length L Ch R = 1 ,24038   ,224.6,232.3,236.2
XS GIS Cut Line= 3
 2232036.2125215414879.8416733762232971.76279822415118.705573813
2233178.28054547415218.232198995
#Sta/Elev= 30
       0 2450.74    20.6 2439.18    74.3 2412.06   116.2 2393.37   132.1 2386.85
   136.2 2386.07   181.6 2382.88   264.1 2381.72   499.5 2381.68   656.4  2380.3
   689.4 2378.35   735.4 2379.75   776.1 2378.17     838 2379.31   852.92378.227
   875.2 2376.04   883.4 2376.02   891.7 2376.05   897.52378.153   899.9 2378.98
   908.2 2378.79   912.3 2379.86   928.8  2390.2   937.1 2391.35   945.3 2395.04
   974.9 2403.84  1027.6 2416.07  1054.8 2421.28  1112.5 2430.33  1194.8 2441.53
#Mann= 6 ,-1,0
       0      .1       0     110     .06       0     210     .05       0
   852.9    .045       0   897.5     .05       0     920      .1       0
Bank Sta=852.9,897.5
XS Rating Curve= 0 ,0
Exp/Cntr(USF)=0,0
Exp/Cntr=0.3,0.1

Type RM Length L Ch R = 1 ,23806   ,500.4,506.8,512.8
XS GIS Cut Line= 3
2232036.56373455415026.9103765732232313.44172449415065.113059833
2233074.87955317415442.990921381
#Sta/Elev= 30
       0 2440.13    80.4 2396.07   100.6  2386.8   108.6 2384.08   112.7 2383.74
   124.8 2383.71     153 2381.84   376.3 2380.31   478.6 2380.58   558.6 2378.94
     773 2379.39     786 2377.53   794.9 2375.81   818.4 2375.25   831.8 2375.99
   839.7 2377.93   845.2 2382.54   854.1 2392.19   867.5 2402.57   898.8 2418.88
     930 2430.51   953.1 2436.07     968 2437.96   983.6 2438.57     997 2437.98
  1014.9 2434.32  1019.4  2434.6  1036.6 2441.23  1081.4 2455.34  1129.5 2469.04
#Mann= 8 ,-1,0
       0      .1       0      10     .06       0     200     .05       0
   299.5      .1       0   309.5     .05       0   749.5      .1       0
     786    .045       0   839.7      .1       0
Bank Sta=786,839.7
XS Rating Curve= 0 ,0
Exp/Cntr=0.3,0.1
